HEC-RAS study SANDRN1.prj: SANDRN1

--- SANDRN1.g01 (geometry) --- (continued)

Type RM Length L Ch R = 1 ,55291   ,55.3,53.9,53.6
XS GIS Cut Line= 4
2207335.43859831705751.9755270572207396.59904749705778.187148136
2207772.29894962705988.9722676442207919.73931819706047.948415071
#Sta/Elev= 30
       0 1676.01    10.6 1672.57    31.3 1669.14      40 1665.97      64 1658.49
    71.4 1654.35    75.2 1652.79    77.2  1652.5   107.3 1652.01   241.8 1654.15
   252.5 1653.77   256.1  1652.8   259.4 1651.74   263.3 1651.46   267.9 1651.73
   270.81652.822     277 1654.28   309.4 1653.88   415.1 1654.81   478.8 1658.18
   497.4 1659.78   514.4  1662.2     562 1667.28   598.9 1670.52   613.5 1670.26
   617.8 1671.46   622.1 1673.71   626.4 1674.62   639.4  1675.8   656.1 1676.49
#Mann= 4 ,-1,0
       0     .05       0   256.1    .045       0   270.8     .05       0
  547.33     .06       0
Bank Sta=256.1,270.8
XS Rating Curve= 0 ,0
Exp/Cntr(USF)=0,0
Exp/Cntr=0.3,0.1

Type RM Length L Ch R = 1 ,55237   ,694.7,707.9,703.9
XS GIS Cut Line= 4
2207305.95052459705800.030165702 2207366.0188229705828.426088537
2207735.16581976706023.9210957492207919.73931819706100.371657229
#Sta/Elev= 30
       0 1682.43    11.3 1678.62    24.6 1676.28    33.4  1671.8    58.8 1663.88
    64.4 1661.28    73.4 1654.24    77.9 1652.77   109.6 1651.72   141.3 1652.99
   221.9 1652.98   236.4 1653.49   245.4 1652.64   249.1 1651.61     268 1650.65
  273.38 1651.59   278.7 1653.15   286.1 1653.75   368.1 1653.87   397.1 1653.38
   461.2 1655.25   493.9 1659.29   558.9 1665.09   584.8  1667.9     602 1669.01
   619.5 1671.25   636.8  1671.5   645.4 1676.82   662.8 1678.49   683.9 1683.37
#Mann= 4 ,-1,0
       0     .05       0   249.1    .045       0  273.38     .05       0
  574.16     .06       0
Bank Sta=249.1,273.38
XS Rating Curve= 0 ,0
Exp/Cntr(USF)=0,0
Exp/Cntr=0.3,0.1

Type RM Length L Ch R = 1 ,54529   ,835.8,865.2,861.9
XS GIS Cut Line= 4
2206763.63573183706214.4286805392206941.74904379706249.385498776
2207562.64872008706563.9968629012207880.58930499706585.636797999
#Sta/Elev= 30
       0 1725.63    19.8 1718.62    86.2 1699.35   183.2  1668.4   202.2 1658.84
   224.8 1652.88     256 1651.35   313.8 1651.91   368.1 1650.66   414.7 1652.11
   421.9  1651.6   426.4 1650.15   433.2 1649.08  437.871650.206   448.8 1652.12
   489.2 1650.92   560.9 1650.81   785.1 1653.09   811.1 1653.94   838.9 1656.79
   899.1 1660.76   903.2 1662.18   915.2  1671.5   923.2 1676.09   947.3  1685.1
   992.7 1705.24  1015.2 1712.92  1091.6 1734.33  1154.1 1758.53  1196.2 1770.92
#Mann= 7 ,-1,0
       0      .1       0  281.51     .05       0   426.4    .045       0
  437.87     .05       0  831.51     .08       0  861.51     .06       0
 1137.57      .1       0
Bank Sta=426.4,437.87
XS Rating Curve= 0 ,0
Exp/Cntr(USF)=0,0
Exp/Cntr=0.3,0.1

Type RM Length L Ch R = 1 ,53664   ,749.7,759,757.2
XS GIS Cut Line= 4
2206690.28385648706632.3170221762206783.50203844706717.212152178
 2207004.8952206 707241.564425722207074.80885708707434.659231215
#Sta/Elev= 30
       0 1711.54    33.1 1695.94    52.9 1688.11    64.2 1685.87    75.6 1681.33
   129.6 1662.95   147.9 1658.65   199.8 1650.84   208.5 1650.32   304.1  1650.5
   340.3 1649.15   389.1 1650.36   395.3  1649.8   403.9 1648.17   408.3 1648.26
  414.06 1649.81   477.5 1649.86   503.8  1655.3   521.2 1657.08   535.7 1657.18
   538.5 1657.89   542.9 1661.06   547.2 1662.57   564.6 1663.84   581.5  1667.8
     615 1677.51   655.8 1685.39   686.2 1688.58   792.7 1696.73   900.6 1706.71
#Mann= 6 ,-1,0
       0      .1       0  246.08     .05       0   395.3    .045       0
  414.06     .05       0  486.08     .06       0  596.08     .05       0
Bank Sta=395.3,414.06
XS Rating Curve= 0 ,0
Exp/Cntr(USF)=0,0
Exp/Cntr=0.3,0.1

Type RM Length L Ch R = 1 ,52904   ,551.4,566.4,532.1
XS GIS Cut Line= 3
2206136.11533557706842.6944278112206219.49259487707316.336913827
2206293.53107241707615.391897899
#Sta/Elev= 30
       0 1739.18    26.4 1725.03    51.3 1709.38    63.4 1700.96    95.9 1681.14
   119.6 1669.22   136.6  1661.6   156.9  1656.4   233.6 1648.49   246.2    1648
     275 1648.61   290.9 1646.74  306.59 1648.67   323.4 1649.91   331.5 1649.17
   339.6 1647.45   351.8 1646.93   380.2 1648.43   392.4 1648.22   416.6 1651.53
     433 1653.09   576.6 1660.53   675.5 1669.61   683.7 1672.52   708.4 1668.62
   720.8 1669.58   733.2  1668.5   741.4 1673.56   743.1  1673.8     789 1676.06
#Mann= 6 ,-1,0
       0      .1       0     210     .05       0     275    .045       0
  306.59     .05       0  610.93     .06       0  710.93     .05       0
Bank Sta=275,306.59
XS Rating Curve= 0 ,0
Exp/Cntr(USF)=0,0
Exp/Cntr=0.3,0.1

Type RM Length L Ch R = 1 ,52338   ,183.1,187.3,178
XS GIS Cut Line= 5
2205693.93120334706897.8723091182205770.38176482706994.952387191
2205930.56389364707412.3967229032206003.37395219707554.376337084
2206050.70049025707649.029413205
#Sta/Elev= 30
       0 1691.87    26.7 1680.46    74.7  1661.3    89.4 1656.53   179.3 1649.18
   210.3 1647.36   228.8  1645.9   242.5 1647.39   272.2 1647.55   310.2 1648.84
   365.9 1647.53   464.4 1648.22   482.8 1649.76     503 1652.74   541.5 1654.72
   560.2 1655.07     583 1654.29   643.8 1657.68   661.9    1658   688.4 1663.13
   737.9 1667.58   746.8 1667.86   759.8 1667.01   773.6 1667.82   782.6 1667.39
   787.1 1669.33   791.5 1672.23     796 1673.87   809.4 1675.35   836.1 1680.55
#Mann= 6 ,-1,0
       0      .1       0  183.57     .05       0   210.3    .045       0
   242.5     .05       0  720.69     .06       0  830.25     .05       0
Bank Sta=210.3,242.5
XS Rating Curve= 0 ,0
Exp/Cntr(USF)=0,0
Exp/Cntr=0.3,0.1

Type RM Length L Ch R = 1 ,52151   ,66.7,66.5,66.4
XS GIS Cut Line= 4
2205615.68828227706973.5964476482205626.60979105707057.692065276
2205877.80449306707460.6957393612205918.21407555 707550.25211138
#Sta/Elev= 30
       0 1673.42    11.7 1669.28    23.8 1665.65    39.9 1659.79    98.3 1655.01
   131.3 1651.23   155.3  1650.5   187.2    1648   216.2  1647.5   219.1 1647.02
   223.9  1645.6   230.3 1644.39     235 1644.75   239.7 1645.59   249.2 1647.63
   256.9 1648.24   272.7 1648.35   291.9 1647.72   362.3 1648.52   381.1 1648.42
   404.7  1648.9   423.6 1648.76   451.4 1649.07   461.3 1649.65   496.1 1650.51
   508.4 1651.39   533.9 1654.26   573.4 1657.71   604.3 1660.86   657.9  1665.2
#Mann= 5 ,-1,0
       0      .1       0   194.8     .05       0   223.9    .045       0
   239.7     .05       0   544.8     .06       0
Bank Sta=223.9,239.7
XS Rating Curve= 0 ,0
Exp/Cntr(USF)=0,0
Exp/Cntr=0.3,0.1

Type RM Length L Ch R = 1 ,52084   ,656.8,680.5,662.7
XS GIS Cut Line= 4
2205548.18384924706994.6281037572205561.28965978707079.815872262
2205816.85296529707485.0038481042205859.44684955707562.546560462
#Sta/Elev= 30
       0 1663.78     7.8 1662.32    26.8 1659.85    51.1 1657.88    75.4 1654.74
   121.2 1651.09   172.9 1648.45   187.9 1648.63     214 1647.53   229.7 1647.64
  235.671645.771   239.1 1644.83   248.6 1644.71   254.6 1645.72   258.1 1646.74
     294 1648.01   366.8 1647.55   414.3 1647.66   437.3 1648.11   466.3 1650.22
   496.5  1653.2     504 1653.56   527.6 1653.18     549 1654.61     564 1656.21
   574.6 1654.85   588.4 1654.28   614.9  1656.7   638.6 1662.24   653.7 1665.07
#Mann= 5 ,-1,0
       0      .1       0  235.67    .045       0   254.6      .1       0
  256.19     .05       0  516.19     .06       0
Bank Sta=235.67,254.6
XS Rating Curve= 0 ,0
Exp/Cntr(USF)=0,0
Exp/Cntr=0.3,0.1

Type RM Length L Ch R = 1 ,51404   ,526.1,532.9,537.5
XS GIS Cut Line= 4
2204993.77040717707099.7558215932205085.84874668707229.229657362
2205314.58751695707531.4121680792205390.29787575707796.074135175
#Sta/Elev= 30
       0 1718.29    14.2 1716.45    45.6 1705.58    77.3 1689.48   114.6 1672.24
   168.8 1651.11   182.6 1649.01   217.6 1646.03   235.6 1646.78     249 1644.06
   259.1 1645.52   264.2 1644.52   274.2 1643.13   284.2 1644.53   289.2 1646.56
   294.3 1646.92   360.4 1646.62   394.3 1648.59   421.2 1647.06   476.9 1648.71
   560.5 1660.07   595.6  1666.7   631.2 1669.13   647.9 1672.87   664.5 1672.87
   672.8 1678.01   731.4  1703.1   764.4 1711.95   797.7 1716.33   813.1 1719.74
#Mann= 5 ,-1,0
       0      .1       0   264.2    .045       0   284.2     .05       0
  657.87     .06       0  757.87      .1       0
Bank Sta=264.2,284.2
XS Rating Curve= 0 ,0
Exp/Cntr(USF)=0,0
Exp/Cntr=0.3,0.1

Type RM Length L Ch R = 1 ,50871   ,381.3,365.7,339.1
XS GIS Cut Line= 4
2204576.04716094 707054.526536212204617.30619412707254.754197234
2204721.66727804 707783.840622732204846.84265032707966.749677234
#Sta/Elev= 30
       0 1767.57    23.1 1762.56    55.8 1749.79    84.4 1740.19   141.6 1734.17
   190.6 1722.78     211  1714.7     260 1689.45   276.2 1682.39   280.5 1680.12
   292.5  1670.8   296.6 1669.09   321.1 1667.19   334.9 1660.39   345.5 1656.88
   353.7 1654.96     370 1654.31   382.2 1645.08   392.31642.938   398.5 1641.99
   409.9 1642.91     423 1644.94   439.3 1645.42   533.1 1644.91     635  1646.5
   695.9 1649.05     741 1652.72   803.5 1654.29   847.1 1657.44   965.4 1662.57
#Mann= 6 ,-1,0
       0      .1       0     200     .05       0   392.3    .045       0
   409.9     .05       0  813.72     .07       0  933.72     .08       0
Bank Sta=392.3,409.9
XS Rating Curve= 0 ,0
Exp/Cntr(USF)=0,0
Exp/Cntr=0.3,0.1

Type RM Length L Ch R = 1 ,50505   ,41.2,42.3,44
XS GIS Cut Line= 6
2204263.93621866707699.6228115632204544.38977753707694.229473893
2204653.60486536707947.7163444082204691.35822905707996.256383443
2204745.29160575708007.0430587842204942.14843073708009.739727619
#Sta/Elev= 30
       0 1659.87    12.2 1659.44    28.2 1657.01    68.3 1652.76    96.3 1650.88
   112.3 1648.65   164.3 1646.93   196.3 1644.75   206.7 1642.75   212.3 1641.79
   224.3 1641.49   232.3 1642.78   244.3 1644.98   276.3 1646.79   355.4 1646.54
   375.2 1645.21     410 1647.81   527.6 1647.78   593.8 1647.04     618 1647.66
   643.4 1649.81   670.5 1650.63   747.7 1660.68   768.2 1662.14   800.4 1665.71
   816.5 1665.75   820.5 1667.17   844.7 1681.54   860.8 1684.88   870.8 1687.73
#Mann= 7 ,-1,0
       0     .06       0   206.7    .045       0   232.3     .06       0
  550.51     .05       0  576.52      .1       0  693.01     .08       0
  787.74     .07       0
Bank Sta=206.7,232.3
XS Rating Curve= 0 ,0
Exp/Cntr(USF)=0,0
Exp/Cntr=0.3,0.1

Type RM Length L Ch R = 1 ,50463   ,430.3,423,407
XS GIS Cut Line= 6
2204278.76789725707731.9828375872204517.42308917707737.376175257
2204654.95319977708017.8297341252204735.85326483708047.493091313
2204818.10166431708040.7514192242204950.23843723708047.493091313
#Sta/Elev= 30
       0 1662.25    14.3 1663.47    41.4 1663.19    53.4 1661.44    65.4  1661.2
    97.4 1656.49   129.4 1649.67   169.5 1647.75   185.5 1646.28   197.5 1644.08
   205.5 1642.01   217.5 1641.78   225.4 1642.49   229.5 1644.06   229.5 1644.07
   238.7 1645.48   328.5  1644.3   446.9  1644.9     519 1646.44   552.4 1646.42
   650.9  1649.9   701.8 1654.77   725.9 1658.94     762 1664.14     786 1665.01
   789.7 1666.75     798 1672.75     802 1674.96   821.1 1680.78   852.1 1691.47
#Mann= 7 ,-1,0
       0     .06       0   197.5    .045       0   229.5     .07       0
  348.72     .06       0  458.72     .05       0  561.12      .1       0
  767.66     .06       0
Bank Sta=197.5,229.5
XS Rating Curve= 0 ,0
Exp/Cntr(USF)=0,0
Exp/Cntr=0.3,0.1

Type RM Length L Ch R = 1 ,50040   ,600.2,611,612.1
XS GIS Cut Line= 4
2204514.95195717708190.5939388152204602.02032533 708146.17561351
2204733.48880458708070.9255846892204952.77023403708065.195905344
#Sta/Elev= 30
       0 1696.17    23.8 1684.57    46.6 1674.53    64.2 1667.77    86.7 1660.35
   117.6 1652.04   126.4 1650.24   137.1 1649.13   146.3 1644.01   149.81642.679
   155.7 1641.17   161.6 1641.01   183.2 1641.16     1911642.627     197 1644.68
   220.1 1646.12   234.9 1649.15     241 1649.88   299.9 1652.43   355.9 1655.66
   361.1 1656.88   374.4 1662.73     380 1664.35     388 1665.14     400 1665.24
     404 1666.06     412 1671.54     416 1673.67     436 1680.15   468.6 1691.99
#Mann= 4 ,-1,0
       0      .1       0   149.8    .045       0     191      .1       0
  379.23     .06       0
Bank Sta=149.8,191
XS Rating Curve= 0 ,0
Exp/Cntr(USF)=0,0
Exp/Cntr=0.3,0.1

Type RM Length L Ch R = 1 ,49429   ,416.4,416.3,415.3
XS GIS Cut Line= 3
2204564.39206972708619.0650059732205002.12295063 708469.04456322
2205111.04190221708438.218444846
#Sta/Elev= 30
       0 1700.97    54.8 1682.73   135.1 1659.58     143 1655.85   147.8 1654.62
     152 1652.22   160.4 1642.58   164.7    1640   168.9 1639.02   177.4  1638.9
     184 1639.95   194.3 1642.81   219.6 1644.16   270.4 1645.31   309.9 1644.38
   328.8  1644.9   366.6 1650.78   401.5 1659.31   414.2 1661.25   422.6 1664.19
   432.7 1665.78   443.8 1671.86     448 1673.43   461.1 1675.06     494 1687.89
   527.2 1703.83   539.7 1711.23   543.8  1712.3   564.5 1714.21   575.9  1716.6
#Mann= 4 ,-1,0
       0      .1       0   164.7    .045       0     184      .1       0
     420     .06       0
Bank Sta=164.7,184
XS Rating Curve= 0 ,0
Exp/Cntr(USF)=0,0
Exp/Cntr=0.3,0.1

Type RM Length L Ch R = 1 ,49013   ,566.8,563.4,557
XS GIS Cut Line= 3
2204765.10224366708940.3030540132205202.83312457708749.181120095
2205342.57819454708662.867988648
#Sta/Elev= 30
       0 1694.62    20.8 1684.03    41.2 1675.49    77.6 1664.89      95 1660.99
     111 1654.93   144.5 1646.02   171.8 1643.22   223.5 1644.15   282.7 1643.66
   287.1  1643.3   293.91639.832   304.5 1638.48   315.41640.292   326.3 1645.88
   341.9  1660.7     348 1664.98   365.6 1665.91   374.3 1671.18   378.4 1672.58
   404.9 1678.73     430 1690.46   445.2  1692.2   464.7 1702.15   481.5 1708.26
   492.9 1710.16   516.8 1716.42   549.7 1721.69   609.4 1740.55   641.9 1749.14
#Mann= 6 ,-1,0
       0      .1       0     110     .05       0   293.9    .045       0
   315.4     .05       0     430     .06       0  537.64      .1       0
Bank Sta=293.9,315.4
XS Rating Curve= 0 ,0
Exp/Cntr(USF)=0,0
Exp/Cntr=0.3,0.1

Type RM Length L Ch R = 1 ,48449   ,712.7,735.5,755.6
XS GIS Cut Line= 3
2205032.34646377709490.5897524552205373.59159417709187.630661077
2205418.53607475709032.821894604
#Sta/Elev= 30
       0 1699.48    10.5 1696.45    37.7 1686.74    85.4 1670.95   131.2 1656.91
     151 1649.84   182.2 1642.48   202.1 1641.17   208.81640.034   216.2 1638.44
   229.41639.292   244.6 1641.13   277.9 1641.93   309.7 1643.76   338.1 1647.07
   352.8 1650.76   363.5 1651.34   369.2 1650.84   372.1 1651.38   374.9 1652.85
   383.4 1660.21   386.2 1661.95   431.6 1677.14   448.6 1683.54   465.6 1691.05
   492.2  1704.4   517.2 1714.58   534.6 1720.11   550.5 1723.63   617.5 1732.38
#Mann= 4 ,-1,0
       0     .05       0   208.8    .045       0   229.4     .05       0
     430     .06       0
Bank Sta=208.8,229.4
XS Rating Curve= 0 ,0
Exp/Cntr(USF)=0,0
Exp/Cntr=0.3,0.1

Type RM Length L Ch R = 1 ,47714   ,117.2,117.9,118.5
XS GIS Cut Line= 3
2205205.98843134709758.7991031842205465.16826941710031.462285424
2205567.04242541710103.373454367
#Sta/Elev= 30
       0  1691.5    25.4 1678.58    36.4 1672.43      53 1665.51    80.5 1652.99
    90.9  1648.9   101.9 1645.89   113.5 1644.17     139  1642.5   198.5 1641.64
   232.4 1640.41   246.1 1638.98   253.31637.443   258.6  1636.6   268.2 1636.73
     272 1637.38   277.7 1639.76     289 1645.98   293.5 1647.52   311.6  1648.2
   325.8 1653.23     351 1658.04   363.1 1661.18   379.2 1663.73   404.4 1668.88
     419 1673.01   443.5 1679.07   453.3 1680.83     468 1684.54   500.9 1691.18
#Mann= 6 ,-1,0
       0      .1       0     220     .05       0   253.3    .045       0
     272     .05       0     340     .06       0     360      .1       0
Bank Sta=253.3,272
XS Rating Curve= 0 ,0
Exp/Cntr(USF)=0,0
Exp/Cntr=0.3,0.1

Type RM Length L Ch R = 1 ,47596   ,40.7,41.7,42.4
XS GIS Cut Line= 3
2205171.82302432709883.3660630062205378.23954031710113.809898324
2205427.38632984710207.734873857
#Sta/Elev= 30
       0 1661.74    18.5 1653.66    23.9 1651.83    42.5 1646.19    52.5 1644.62
    84.5 1644.65    93.7 1642.75    99.1 1642.32   185.7 1640.42   192.4 1639.82
   199.8 1637.81   206.5 1636.47   216.8 1636.87  221.571637.772   233.3 1642.65
   236.6 1643.15     248 1643.35   256.5 1641.86   259.3 1642.14   276.3 1646.72
     287  1650.2   297.8 1652.68   316.3 1658.04   322.2 1660.15   340.3  1667.8
   354.8 1674.42   362.8 1678.68   369.6 1680.58   399.8 1692.76   415.4 1698.35
#Mann= 5 ,-1,0
       0      .1       0     160     .06       0   199.8    .045       0
  221.57     .06       0     290      .1       0
Bank Sta=199.8,221.57
XS Rating Curve= 0 ,0
Exp/Cntr(USF)=0,0
Exp/Cntr=0.3,0.1

Type RM Length L Ch R = 1 ,47554   ,209.7,219.8,228.6
XS GIS Cut Line= 3
2205149.98000675 709906.301231452205335.64565606710133.468614133
2205382.60814383710224.117137031
#Sta/Elev= 30
       0 1661.29    19.2 1652.82    39.9 1645.21    50.2  1642.5    63.3 1642.16
    79.3 1641.17   100.3 1641.58     138 1641.57     160 1640.29   184.5 1640.97
   194.9  1639.6  200.581637.985   205.4 1636.33   210.4 1635.75   218.4  1636.2
   222.5 1637.09   224.7 1637.96     231 1642.48   233.9 1643.62   236.7 1644.27
   245.2 1644.75   256.9 1644.62     268 1648.68   302.1 1658.07   311.9  1661.3
   333.6 1669.82   342.6 1673.94   360.6 1683.08   378.7 1690.99   395.5 1696.35
#Mann= 5 ,-1,0
       0      .1       0     170     .06       0  200.58    .045       0
   224.7     .06       0  333.39      .1       0
Bank Sta=200.58,224.7
XS Rating Curve= 0 ,0
Exp/Cntr(USF)=0,0
Exp/Cntr=0.3,0.1

Type RM Length L Ch R = 1 ,47334   ,696.4,658.1,632.1
XS GIS Cut Line= 4
 2205034.5357987709918.3673081632205054.76081496709995.222369971
2205097.90751633710268.9342567582205147.79588978710303.990951617
#Sta/Elev= 30
       0 1682.16    19.5 1673.84    44.3 1661.32    60.8 1654.18    69.1 1649.53
    73.2 1647.88    77.4    1647    93.6 1645.74   105.7 1643.35     130 1640.89
   142.2 1640.35   169.9 1640.62   183.9 1640.09   190.8 1639.47  195.861638.016
   202.9 1636.08   218.8 1635.43   223.2 1635.59   227.2 1636.69   229.1 1638.01
   236.3 1642.04   243.4 1644.46   251.5 1644.13   320.4 1646.63   328.5 1647.92
   344.8 1651.73   358.4 1652.67     374  1655.1   393.6 1656.55   417.5 1657.32
#Mann= 5 ,-1,0
       0      .1       0  189.47     .05       0  195.86    .045       0
   229.1     .05       0  406.56     .06       0
Bank Sta=195.86,229.1
XS Rating Curve= 0 ,0
Exp/Cntr(USF)=0,0
Exp/Cntr=0.3,0.1

Type RM Length L Ch R = 1 ,46676   ,639.3,608.6,584.7
XS GIS Cut Line= 4
2204092.12860042710398.1047235882204417.87574633710163.958225028
2205017.01426161710249.7492747392205093.91941506710307.032831348
#Sta/Elev= 30
       0 1782.38    54.2 1774.21   145.5 1758.58   172.5 1752.61   218.5 1737.85
   252.9 1720.42   268.9 1707.43   290.2 1704.25   301.6 1699.34     335  1688.3
   341.8 1685.22   349.8 1680.14   359.7 1677.29   371.7 1670.02   407.2 1651.67
   411.6 1646.13   415.6 1639.61  418.23 1636.97   423.7 1634.61   447.9 1634.47
     452 1634.73   459.4 1636.99   472.2 1639.49   480.3 1639.89     581 1638.99
     650 1641.64     949 1641.89  1006.1 1644.42    1059 1648.24  1102.3  1653.8
#Mann= 8 ,-1,0
       0      .1       0     220     .06       0  418.23    .045       0
   459.4      .1       0  551.17     .05       0  641.17      .1       0
  651.17     .05       0 1086.42     .06       0
Bank Sta=418.23,459.4
XS Rating Curve= 0 ,0
Exp/Cntr(USF)=0,0
Exp/Cntr=0.3,0.1

Type RM Length L Ch R = 1 ,46067   ,442.9,425.3,396.8
XS GIS Cut Line= 3
2204721.30830663 710756.164294262204827.24694183710629.474792376
2205028.20270344710355.344921919
#Sta/Elev= 30
       0 1712.42     4.5 1711.32    19.5 1704.95      24 1703.74    29.7 1703.13
    38.2 1700.53    73.1 1687.95   114.9 1671.57   134.2 1662.75   149.9  1658.1
   154.7 1655.78   160.3  1651.6   180.4 1650.54   190.3 1646.42   200.5  1643.2
   223.3 1638.97   240.4 1637.72   274.6 1638.44   283.4 1636.09   289.1 1634.75
     302 1634.12   306.2 1634.39     312 1636.11   320.6 1638.68   329.1 1639.56
   362.9 1640.41   373.8 1640.17   426.4 1642.97     473 1643.99     505 1646.66
#Mann= 6 ,-1,0
       0     .05       0      90      .1       0  215.15     .06       0
   283.4    .045       0     312     .06       0  345.15     .05       0
Bank Sta=283.4,312
XS Rating Curve= 0 ,0
Exp/Cntr(USF)=0,0
Exp/Cntr=0.3,0.1

Type RM Length L Ch R = 1 ,45642   ,33.5,35.4,37.3
XS GIS Cut Line= 6
2205189.29743837711021.3872781772205279.94596127710896.882078053
2205249.36573668710820.4315165732205045.13352244710614.015000578
2205037.48846629710552.8545513942205091.00385932 710408.69063546
#Sta/Elev= 30
       0 1690.86    16.5  1684.8    30.8 1677.72    54.7 1667.57    74.5 1660.86
    89.3 1654.87   113.9 1646.89     154 1641.35   201.1 1640.08   209.7 1639.45
   243.8 1641.31     265 1641.49   268.6 1640.72   274.2  1637.5   285.3 1632.88
     290 1631.96   301.5  1631.8   307.5 1631.98   310.7  1632.9   324.1 1636.79
   330.4 1639.28   335.2 1640.08   340.7 1640.31   403.6 1638.76   489.5 1638.76
   526.8 1638.15   585.7 1639.49   671.2 1642.33   711.6 1644.27   742.2 1646.58
#Mann= 8 ,-1,0
       0      .1       0  174.01     .05       0  234.01      .1       0
   285.3    .045       0   310.7     .06       0  556.79     .05       0
  648.42      .1       0  658.42     .05       0
Bank Sta=285.3,310.7
XS Rating Curve= 0 ,0
Exp/Cntr(USF)=0,0
Exp/Cntr=0.3,0.1

Type RM Length L Ch R = 1 ,45607   ,498.7,528.2,558.5
XS GIS Cut Line= 6
2205225.33841735711030.1244852032205320.35554376710895.789927175
2205269.02445249710797.4963481292205089.91170845710582.342625108
2205081.17450142710539.7487408542205118.30763128710425.072898635
#Sta/Elev= 30
       0  1676.9    19.9  1668.9    53.4 1657.33    84.4 1648.56     106 1644.35
   122.7 1642.91   140.5 1638.93   143.4 1638.57   162.8 1639.81   205.1 1639.95
   291.5 1641.76   295.5 1640.61   301.8 1637.55  313.851633.134   317.5 1631.82
   322.7 1631.34   333.1 1631.85   335.9 1633.14   343.5 1636.22   350.1 1637.77
   359.1 1640.77   370.5 1640.77   400.8 1638.05   473.6 1639.38   495.6 1640.52
   555.4 1641.17   639.4 1645.94   660.5 1648.59   706.7 1651.46   719.4 1652.82
#Mann= 7 ,-1,0
       0      .1       0  184.54     .05       0  295.43     .06       0
  313.85    .045       0   335.9     .06       0  545.43      .1       0
  648.86     .05       0
Bank Sta=313.85,335.9
XS Rating Curve= 0 ,0
Exp/Cntr(USF)=0,0
Exp/Cntr=0.3,0.1

Type RM Length L Ch R = 1 ,45079   ,365.7,371.1,380.6
XS GIS Cut Line= 4
2205244.74982521711068.8959553592205325.64989027711062.154283271
2205509.02337108710994.7375623872205631.72180309711002.827568893
#Sta/Elev= 30
       0 1670.96    23.5 1660.98    55.6 1649.55    75.7 1645.17    79.7 1643.85
    83.9 1641.68    88.1 1641.02   100.9 1641.45   107.2  1640.3   109.4 1639.41
     118 1632.94   121.3 1631.48   126.5 1630.25     135 1630.01   147.8 1630.14
   152.1 1630.78   153.6  1631.5   158.7 1634.04   161.8 1634.89   228.8 1637.63
   241.6 1638.39   258.6 1640.58   271.4 1640.68   303.8 1646.03   323.8 1647.35
   355.9 1656.54   374.5  1663.9   387.9  1672.4     396 1673.39   399.5 1674.46
#Mann= 5 ,-1,0
       0      .1       0   121.3    .045       0   153.6      .1       0
  221.18     .06       0  316.55      .1       0
Bank Sta=121.3,153.6
XS Rating Curve= 0 ,0
Exp/Cntr(USF)=0,0
Exp/Cntr=0.3,0.1

Type RM Length L Ch R = 1 ,44708   ,604.2,597.8,588
XS GIS Cut Line= 4
2205177.84446298711379.5370842962205249.42270984711381.201694688
2205605.64933377711374.5432531192205753.79965868 711344.58026606
#Sta/Elev= 30
       0 1685.48    62.3 1660.32    78.4 1655.94    82.4 1653.94    90.4 1647.63
   106.4 1647.08   138.4 1634.85   146.4 1634.64   155.9 1636.75   182.4 1637.11
   246.4 1634.89   250.4 1635.76   282.4 1635.13   310.4 1633.32   317.8 1630.44
   322.4 1628.71   333.5 1628.54   346.4 1628.74   354.4 1630.58   362.4 1636.19
   370.4 1645.55   374.4 1649.07   390.4 1657.71     438 1670.48   475.1 1687.34
   499.8 1697.18     508 1698.64   548.8 1711.72   570.4 1715.46     579 1718.08
#Mann= 6 ,-1,0
       0      .1       0   181.6     .06       0   281.6     .05       0
   317.8    .045       0   354.4     .05       0   371.6      .1       0
Bank Sta=317.8,354.4
XS Rating Curve= 0 ,0
Exp/Cntr(USF)=0,0
Exp/Cntr=0.3,0.1

Type RM Length L Ch R = 1 ,44110   ,167,164.6,163
XS GIS Cut Line= 4
2205382.43220951  711908.94585612205445.31749099711925.591960021
2205776.39000233711749.8830852912205878.11619296711651.856028862
#Sta/Elev= 30
       0 1677.29    22.5 1668.69    59.7 1652.24    94.1 1642.63   105.9 1635.86
     109  1635.3   122.6 1635.74   136.2 1633.47   163.4 1631.88  178.511628.388
   182.8 1627.64   194.7 1627.32   200.6 1628.33   206.5 1630.86   217.7 1632.07
   295.3  1632.9     340 1634.93   358.1  1637.2   367.2 1640.16   376.2 1644.59
   380.7 1645.12   389.8 1642.75   404.7 1643.47   432.8  1642.7   445.9 1643.64
   468.5 1650.24   527.9 1663.18   550.5 1670.51   564.7 1674.33   581.1 1680.28
#Mann= 5 ,-1,0
       0      .1       0  178.51    .045       0   200.6     .06       0
  295.05     .05       0  405.05      .1       0
Bank Sta=178.51,200.6
XS Rating Curve= 0 ,0
Exp/Cntr(USF)=0,0
Exp/Cntr=0.3,0.1

Type RM Length L Ch R = 1 ,43945   ,58,59.1,59.1
XS GIS Cut Line= 3
2205319.26339289712198.7259249662205847.86441798711869.988510603
2205940.69724263711762.957724531
#Sta/Elev= 30
       0 1639.84    10.5 1640.06    33.2  1637.7    90.6 1634.37   193.5 1632.59
   236.6 1631.08   251.6 1631.13     269 1632.79   277.7 1632.69   283.2 1631.64
   298.3 1627.15   305.9  1626.3   316.7 1626.78   335.5 1625.97   340.2    1626
   344.9 1626.84   353.2 1629.86   358.9 1630.34   428.7 1630.61   509.8 1632.84
   533.4 1632.07   559.4 1635.05   588.4 1634.78     603 1635.97   634.1  1640.7
   660.1 1643.79   676.5 1647.02   718.9 1658.86   750.6 1671.44   764.2 1676.31
#Mann= 7 ,-1,0
       0     .05       0     250      .1       0     270     .07       0
   316.7    .045       0   344.9     .07       0     390     .05       0
     620      .1       0
#XS Ineff= 2 , 0
          274.34 1651.78
Permanent Ineff=
       F       F
Bank Sta=316.7,344.9
XS Rating Curve= 0 ,0
Exp/Cntr(USF)=0,0
Exp/Cntr=0.3,0.1

Type RM Length L Ch R = 1 ,43886   ,379.1,368.1,360.3
XS GIS Cut Line= 3
2205371.68663504712231.4904513152205893.73475486711910.398093099
2205975.64607073711783.708591219
#Sta/Elev= 30
       0 1642.81    85.1  1638.1     130 1636.58   188.4 1634.37     226 1633.46
   235.4 1633.34   257.9 1634.03   268.2 1632.64   282.3 1629.79   289.9 1629.04
   295.7 1627.26   301.5 1625.98   309.8 1625.76   319.9 1626.07   324.6 1627.31
   330.6    1629   333.5 1629.32   413.8 1629.46   449.8 1630.83     476 1630.23
   521.8 1630.82   557.4 1630.23   568.8 1630.72   623.9 1637.69   641.6 1641.11
   676.3 1649.09   690.6 1653.41   705.2 1658.76   723.9 1667.15   763.8 1678.51
#Mann= 10 ,-1,0
       0     .05       0     100      .1       0     130     .05       0
     210     .07       0   295.7    .045       0   324.6     .07       0
     330     .05       0     440      .1       0     510     .05       0
     560      .1       0
#XS Ineff= 2 , 0
                          456.14         1632.88
Permanent Ineff=
       F       F
Bank Sta=295.7,324.6
XS Rating Curve= 0 ,0
Exp/Cntr(USF)=0,0
Exp/Cntr=0.3,0.1

Type RM Length L Ch R = 1 ,43518   ,891.1,883.4,861.5
XS GIS Cut Line= 4
2205724.39015539712491.7039818312205929.65406965 712294.64831428
2206030.69528636 712107.38708656  2206174.928079711902.838722799
#Sta/Elev= 30
       0  1709.4    10.1 1704.63    38.3 1695.76      94  1682.9   131.8 1668.74
   159.6 1656.41   194.2 1645.18   230.8 1636.79   276.9 1631.76   336.2 1627.45
   345.3 1626.04   358.3 1621.77   374.1 1619.82   386.2 1620.08   392.91621.723
   416.2 1625.71   445.3 1626.45   476.4 1624.15   486.2 1630.08   490.7 1631.19
     500 1630.87   514.3  1627.8   522.9 1627.99   544.1 1635.52   627.3  1635.2
     642 1639.83   657.8 1641.83   671.3 1646.02   703.8 1658.86   747.6 1678.57
#Mann= 3 ,-1,0
       0      .1       0   358.3    .045       0   392.9      .1       0
Bank Sta=358.3,392.9
XS Rating Curve= 0 ,0
Exp/Cntr(USF)=0,0
Exp/Cntr=0.3,0.1

Type RM Length L Ch R = 1 ,42635   ,708.8,731.6,737.9
XS GIS Cut Line= 4
2206666.56619933712724.2480336672206696.52918639712646.344267312
2206636.60321227712222.3680004232206590.16058233712089.032708009
#Sta/Elev= 30
       0 1680.37    24.7 1667.57    50.4 1656.36    76.1 1646.99   104.8 1639.66
   109.6 1637.82   116.7 1633.74   123.7 1628.63   133.1 1617.59   137.2 1613.97
   141.2 1612.51   161.4 1612.26   169.5 1612.84   172.81613.987   177.6 1615.81
   185.6 1616.99   213.9 1618.25   254.3  1618.2   270.5 1616.48   286.7 1618.69
   306.8 1619.35   415.9 1618.56     460 1619.84   508.8 1631.24   528.6 1637.73
   569.5 1654.39   618.8 1678.07   631.5 1682.75   641.7 1685.47   652.8 1686.27
#Mann= 3 ,-1,0
       0      .1       0   137.2    .045       0   172.8      .1       0
Bank Sta=137.2,172.8
XS Rating Curve= 0 ,0
Exp/Cntr(USF)=0,0
Exp/Cntr=0.3,0.1

Type RM Length L Ch R = 1 ,41903   ,504.9,522.7,523.9
XS GIS Cut Line= 4
2206729.48847215712733.2369297852206846.34412169712610.388682841
 2207231.3685054712322.7440070712207258.33519375 712180.41981854
#Sta/Elev= 30
       0 1671.11    38.7 1654.78   106.6 1631.37   149.1  1621.8   191.7 1616.53
   211.7  1615.5   326.6 1616.79   371.6 1614.47   425.5 1613.75   485.7 1614.83
   554.7  1612.9     569 1610.71   581.3 1610.11   594.7 1607.15   599.3 1607.86
   603.3 1610.26     606 1612.82   616.2 1627.22   620.4  1631.8     626 1636.35
   631.8 1639.18     664 1648.08   688.4 1656.08   700.6 1661.45   712.8 1663.21
   737.2 1676.46   753.5 1684.35   765.1 1688.71   782.2 1693.18     795 1694.72
#Mann= 3 ,-1,0
       0      .1       0   581.3    .045       0   603.3      .1       0
#XS Ineff= 2 , 0
          285.26 1651.63
Permanent Ineff=
       F       F
Bank Sta=581.3,603.3
XS Rating Curve= 0 ,0
Exp/Cntr(USF)=0,0
Exp/Cntr=0.3,0.1

Type RM Length L Ch R = 1 ,41380   ,433.3,424.4,413.3
XS GIS Cut Line= 4
2206768.51939822712779.2941242712206861.73758018712716.038929367
2207146.38595724712757.6541891722207382.76063293712754.324968388
#Sta/Elev= 30
       0 1672.16    21.4 1660.97    47.9 1648.63    76.9 1636.57   101.1 1627.72
   115.1 1623.88   159.6 1618.99   191.9 1612.59   204.1 1611.52   208.1 1608.88
   212.1 1605.44     2181603.016   224.3 1601.89   232.4 1601.59   246.8 1601.72
   252.71602.491   260.6 1604.78   268.7 1605.77     297 1605.93   421.9 1611.55
   438.2 1611.97   458.5 1609.72   477.5 1610.72   485.4 1612.14   494.1 1614.61
   526.1  1620.7   554.1 1628.02   592.4  1636.4   606.1 1640.36   636.7 1650.58
#Mann= 3 ,-1,0
       0      .1       0     218    .045       0   252.7      .1       0
Bank Sta=218,252.7
XS Rating Curve= 0 ,0
Exp/Cntr(USF)=0,0
Exp/Cntr=0.3,0.1

Type RM Length L Ch R = 1 ,40956   ,119.5,105.7,94.8
XS GIS Cut Line= 4
2206829.61516877713175.6331061662206976.46405826713155.022415044
2207171.48266368713095.6897648012207424.83739745713015.809442681
#Sta/Elev= 30
       0 1698.35    14.7 1693.68    39.9 1682.54    82.4 1659.02   107.2 1646.92
   117.8 1640.45   123.8  1635.5   139.9  1618.1   156.3  1603.4   160.5 1600.83
   168.9 1599.28   177.3 1598.26     194 1598.13   202.3 1598.47   205.2 1599.36
   210.7 1601.18   227.4 1603.78   248.3 1603.68   264.6 1602.25   290.1 1602.24
   323.6 1603.89   340.3 1603.84   352.9  1606.7   369.6 1604.78   432.5 1605.39
   453.5 1606.31   499.7 1614.49   524.8 1621.61     550 1630.41   617.8 1656.25
#Mann= 3 ,-1,0
       0      .1       0   168.9    .045       0   205.2      .1       0
#XS Ineff= 2 , 0
                          354.44         1610.02
Permanent Ineff=
       F       F
Bank Sta=168.9,205.2
XS Rating Curve= 0 ,0
Exp/Cntr(USF)=0,0
Exp/Cntr=0.3,0.1

Type RM Length L Ch R = 1 ,40850   ,38.9,39.3,38
XS GIS Cut Line= 6
2206936.56621406713348.7308273782206982.76419621713338.901469473
2207021.09869204713275.9935788842207090.88713316713206.205137762
2207236.36163015713132.4849534782207460.47099037713063.679448146
#Sta/Elev= 30
       0 1645.65    36.4 1630.65    47.2 1623.78    65.3 1615.56    86.7 1607.98
    96.1 1605.83   127.9 1603.11   147.5 1600.08   153.5 1598.68   167.5 1598.18
   181.6  1598.2   190.1 1600.18   193.1 1600.97   204.4 1600.51   215.6 1602.17
   221.9 1601.21   252.4 1605.04   256.9 1604.78   265.9 1602.15   286.8 1602.96
   295.7 1604.35     302 1603.11   324.2    1603   334.4 1605.41   354.6 1604.19
   395.5 1604.05   445.3 1607.45   487.1 1617.09   524.8 1628.92   617.1 1666.35
#Mann= 3 ,-1,0
       0      .1       0   147.5    .045       0   190.1      .1       0
#XS Ineff= 1 ,-1
  250.82  295.99 1606.31
Permanent Ineff=
       F
Bank Sta=147.5,190.1
XS Rating Curve= 0 ,0
Exp/Cntr(USF)=0,0
Exp/Cntr=0.3,0.1

Type RM Length L Ch R = 1 ,40811   ,528.6,537.7,536.5
XS GIS Cut Line= 6
2206943.96955457713384.0865773842207022.60441781713366.393733156
2207049.14368415713302.5029067762207113.03451053713236.646208815
2207246.71377803713166.8577676932207460.99378035713107.881620265
#Sta/Elev= 30
       0 1644.27    24.8 1635.32    28.9 1632.89    37.1  1624.9    41.2 1622.07
    57.6 1616.36      74 1613.96    80.6 1608.97    86.2  1606.5   103.6  1604.9
   116.6 1605.92   126.4 1605.16   157.2 1601.04   169.8 1597.96   186.8 1596.51
   211.6 1596.73   223.6 1598.06   234.6 1600.57   255.3 1600.22   296.8 1602.18
   326.3 1601.62   352.8 1606.83   366.9 1604.37   394.9 1603.66   456.1 1603.64
   476.8 1606.29   497.6 1612.34     518 1619.77   563.8  1639.1   614.6 1663.07
#Mann= 3 ,-1,0
       0      .1       0   169.8    .045       0   223.6      .1       0
Bank Sta=169.8,223.6
XS Rating Curve= 0 ,0
Exp/Cntr(USF)=0,0
Exp/Cntr=0.3,0.1

Type RM Length L Ch R = 1 ,40273   ,413.6,419.2,427.1
XS GIS Cut Line= 4
2207147.56768777713809.6572618652207196.71447729713784.537791663
2207450.09348106 713554.093956342207583.33588821713526.790184382
#Sta/Elev= 30
       0 1640.76    15.7 1633.82    53.8 1618.78    60.2 1613.61    65.3 1608.11
    71.3 1600.38    74.2 1597.36      77 1595.15    79.8 1593.89    92.3 1592.87
   113.9 1593.13  120.71 1593.91   125.1 1596.08   130.8 1597.08   156.3 1596.88
   178.8 1597.59   198.8 1596.74   235.6 1596.49   309.9 1597.55   319.4 1596.69
   331.9 1593.96     341 1594.15     346  1595.9   377.2 1616.44   403.9 1625.24
   444.7  1645.1   461.1 1651.06   481.6 1660.11   514.1 1676.69   533.7 1685.98
#Mann= 3 ,-1,0
       0      .1       0    79.8    .045       0  120.71      .1       0
Bank Sta=79.8,120.71
XS Rating Curve= 0 ,0
Exp/Cntr(USF)=0,0
Exp/Cntr=0.3,0.1

Type RM Length L Ch R = 1 ,39854   ,385.3,409.5,435.9
XS GIS Cut Line= 4
2207140.95821666713899.9360898752207536.65101694713852.134275076
2207674.74514858713789.7263501992207694.66257141713597.191262814
#Sta/Elev= 30
       0 1667.98    23.4 1656.49    71.7 1626.49    95.2 1613.29   116.1 1604.67
   140.2 1598.11   273.2 1595.05   329.6 1596.12   402.4  1595.6   433.7 1593.24
     467 1593.27   477.1 1589.99   485.8 1588.42   512.2 1588.66   516.6 1589.86
     521 1594.32   530.4 1609.31   542.9 1620.51   562.7 1622.49   574.8 1619.41
   586.9 1614.44   598.9  1612.5   602.9 1612.93   627.1 1623.99   639.1  1630.8
   667.3 1642.99   687.4 1649.73   707.5 1658.52   723.6 1663.36   743.7  1675.2
#Mann= 3 ,-1,0
       0      .1       0   477.1    .045       0   516.6      .1       0
Bank Sta=477.1,516.6
XS Rating Curve= 0 ,0
Exp/Cntr(USF)=0,0
Exp/Cntr=0.3,0.1

Type RM Length L Ch R = 1 ,39445   ,642.7,625,606.9
XS GIS Cut Line= 4
2207131.52528723713937.0265137782207246.80787994713944.307519634
2207419.12501852714121.4786621162207593.86915905714254.963769465
#Sta/Elev= 30
       0 1671.58    24.7 1666.25    32.7 1663.13    48.7 1654.32    96.8  1623.7
   115.5 1613.98   144.6  1604.6   155.8 1603.07   213.3  1589.3   218.9 1588.51
   261.8 1587.85   289.6 1589.25   323.6 1589.38   339.9 1590.31     406 1591.79
   414.9 1591.34     426 1589.74   459.6 1590.24   471.6 1584.99   480.8 1583.99
   499.9 1584.03   507.1 1584.93     510 1585.85   514.4 1589.22   520.1 1597.48
   526.9 1605.79   535.1 1614.13   545.8 1623.65   551.5 1627.77   582.6 1643.45
#Mann= 3 ,-1,0
       0      .1       0   471.6    .045       0   507.1      .1       0
#XS Ineff= 2 , 0
          404.17 1633.99
Permanent Ineff=
       F       F
Bank Sta=471.6,507.1
XS Rating Curve= 0 ,0
Exp/Cntr(USF)=0,0
Exp/Cntr=0.3,0.1

Type RM Length L Ch R = 1 ,38820   ,367.7,369.3,364.8
XS GIS Cut Line= 4
2207024.32948721 714534.462915422207281.86136098714520.979571243
2207431.52648134714520.9795712432207505.68487432714512.889564737
#Sta/Elev= 30
       0 1662.05    47.9  1631.8    59.9 1622.42    75.9 1607.57      84 1601.18
      92 1593.44     104 1583.88     112 1579.29     124  1575.6     136 1574.77
   152.1 1574.76   164.1 1575.72   172.1 1580.62   176.1 1581.03   188.1 1580.99
   229.4 1583.53   260.2 1584.56   300.2 1582.81   304.2 1582.01   316.2  1584.4
   344.2  1586.1   360.2 1588.79   372.2 1589.02   376.2 1590.79   384.2 1597.28
     388 1599.26   400.2 1604.99   412.2 1609.27   420.3 1613.25   482.1 1650.47
#Mann= 3 ,-1,0
       0      .1       0     124    .045       0   164.1      .1       0
Bank Sta=124,164.1
XS Rating Curve= 0 ,0
Exp/Cntr(USF)=0,0
Exp/Cntr=0.3,0.1

Type RM Length L Ch R = 1 ,38450   ,343.6,332.9,321
XS GIS Cut Line= 4
 2207056.9602433714806.118944336 2207169.1853861714878.289682357
2207381.53987926714853.0185665672207502.01266965714785.960662275
#Sta/Elev= 30
       0 1649.42    13.3 1642.94    30.6 1633.78    68.2 1612.48    79.9 1606.59
   100.1 1597.67   108.4 1592.87     118 1588.67   136.4 1577.41   144.5 1574.76
   152.6 1573.06   187.5 1569.51   200.9 1567.72     217 1568.21     221 1569.59
   229.1 1574.68   234.3 1575.86   281.5 1576.13   293.5 1576.77   313.7 1575.97
   337.9 1576.44   341.9 1576.71   345.9 1577.84   354.9 1581.42   409.8 1585.76
   413.8 1587.59   425.6 1594.86   437.3 1603.23   475.6 1620.89   485.2 1626.81
#Mann= 7 ,-1,0
       0      .1       0      40     .06       0   187.5    .045       0
     221      .1       0  293.43     .06       0  397.28     .07       0
  417.28      .1       0
Bank Sta=187.5,221
XS Rating Curve= 0 ,0
Exp/Cntr(USF)=0,0
Exp/Cntr=0.3,0.1

Type RM Length L Ch R = 1 ,38117   ,100.7,101.1,101.7
XS GIS Cut Line= 2
2207236.52679543715272.3776802822207575.34476241715022.023934447
#Sta/Elev= 30
       0 1615.86    14.5 1608.09    30.6  1598.1    39.2 1594.15    54.3 1585.03
    62.1 1581.39    69.2 1575.99    73.5 1573.98    94.1 1573.29   113.1 1573.85
   142.2 1572.26   147.9 1571.13   158.7 1566.48   166.9 1564.78   176.5 1564.32
   187.9  1564.8  193.251566.495   223.4 1571.13   278.1 1572.89   283.1 1573.52
     293 1576.87     298 1577.75   312.9 1579.11   322.8  1578.8   332.8 1579.92
   348.7 1583.81     371 1591.03   385.3 1596.37   407.4 1606.38   421.3 1609.64
#Mann= 5 ,-1,0
       0      .1       0     110     .06       0   158.7    .045       0
  193.25     .06       0     260      .1       0
Bank Sta=158.7,193.25
XS Rating Curve= 0 ,0
Exp/Cntr(USF)=0,0
Exp/Cntr=0.3,0.1

Type RM Length L Ch R = 1 ,38016   ,39.5,37.6,39.4
XS GIS Cut Line= 3
2207301.05581087715346.1620662592207578.92192947715149.506102661
 2207658.5397285715085.015685448
#Sta/Elev= 30
       0 1613.41    33.2 1594.33    48.9 1586.67    57.5 1581.24    66.1  1574.6
    68.9 1573.11    72.4 1572.42   101.8 1571.67   131.2 1569.75  148.021565.895
   155.7 1564.67   170.4 1564.61   174.8 1564.92     178 1565.84   181.7 1566.55
   204.7 1567.02   237.1 1569.99   255.5 1570.16   268.4 1573.06   278.7 1574.26
     288 1576.11   297.8 1576.77   306.4 1576.57   317.4 1577.81   335.8 1581.61
   364.3  1588.6   372.9 1590.12   389.9 1595.04   429.9 1603.78   442.9 1607.82
#Mann= 4 ,-1,0
       0      .1       0  148.02    .045       0     178     .06       0
     270      .1       0
Bank Sta=148.02,178
XS Rating Curve= 0 ,0
Exp/Cntr(USF)=0,0
Exp/Cntr=0.3,0.1

Type RM Length L Ch R = 1 ,37979   ,340.2,341.5,341.2
XS GIS Cut Line= 3
2207326.53350656 715378.805363862207615.54611703715163.837306486
2207669.68622036715111.289559127
#Sta/Elev= 30
       0 1614.01     9.4  1609.5    29.5 1597.87    51.9 1586.36    56.7  1583.2
      63 1578.01    70.9 1574.18    73.8  1573.4    83.2 1572.39    93.8 1569.97
   126.7  1567.8   136.7  1565.1   150.2 1563.82   165.3 1563.64   176.5 1564.21
   185.3 1563.89   190.4  1565.1   196.5 1566.84   206.4 1566.91   219.6 1569.22
   231.4 1568.82   241.3 1569.11   265.3 1572.26   279.6  1572.8   336.1 1576.96
     351 1581.46   388.9 1595.47   411.2 1601.08   427.2 1606.15   435.6 1608.27
#Mann= 5 ,-1,0
       0      .1       0     120     .06       0   136.7    .045       0
   190.4     .06       0     240      .1       0
Bank Sta=136.7,190.4
XS Rating Curve= 0 ,0
Exp/Cntr(USF)=0,0
Exp/Cntr=0.3,0.1

Type RM Length L Ch R = 1 ,37637   ,797.3,790.5,771.2
XS GIS Cut Line= 5
2207450.43058747715636.9358465642207561.20036091715626.293899121
2207732.44165264715480.486091467 2207800.7295616715245.961828089
2207777.49693938715143.925416726
#Sta/Elev= 30
       0 1618.64    29.9 1600.96    41.9 1592.31      54 1591.81    70.1 1593.88
   102.2 1595.11   128.4 1592.95   136.9 1591.06   142.6 1587.82   146.7 1584.29
   151.1  1579.4   159.6 1567.22   162.4 1564.16   167.7  1561.1   179.4 1559.46
   190.8 1559.54   202.1 1561.08   233.4 1564.76   298.1 1562.17   335.1 1564.84
   385.5  1563.8   410.5 1564.43   435.4 1567.44   568.8 1567.04   577.1 1568.53
   593.6 1568.94   618.2 1572.66   626.4 1574.88   645.1 1582.67   685.1 1602.99
#Mann= 5 ,-1,0
       0      .1       0  141.28     .06       0   167.7    .045       0
   202.1     .06       0  291.28      .1       0
#XS Ineff= 2 , 0
                          334.73         1566.52
Permanent Ineff=
       F       F
Bank Sta=167.7,202.1
XS Rating Curve= 0 ,0
Exp/Cntr(USF)=0,0
Exp/Cntr=0.3,0.1

Type RM Length L Ch R = 1 ,36847   ,781.3,785.1,785.1
XS GIS Cut Line= 3
 2208196.5264808715787.7587724692208346.19160116715392.696788092
2208424.39499739715257.863346325
#Sta/Elev= 30
       0 1614.15     2.8 1612.54    44.2  1580.1    62.6 1567.13      78 1559.02
      84 1557.29     114 1555.39   156.7    1556   168.4 1551.02   186.7 1549.59
   197.2 1551.12   203.8  1552.3   216.6 1552.18   233.7 1554.18   259.4 1555.03
   293.6 1554.12   310.7 1551.54   323.6 1551.53   327.8 1552.16   332.1  1554.2
     345  1557.6   366.3 1558.46     392  1561.7   404.8 1565.18   413.4 1566.53
   431.2 1572.43     519 1605.82   543.6 1613.93   560.6 1621.05   578.3 1625.99
#Mann= 5 ,-1,0
       0     .07       0      30     .06       0      90      .1       0
   168.4    .045       0   197.2      .1       0
Bank Sta=168.4,197.2
XS Rating Curve= 0 ,0
Exp/Cntr(USF)=0,0
Exp/Cntr=0.3,0.1

Type RM Length L Ch R = 1 ,36061   ,148.2,143.6,141.3
XS GIS Cut Line= 4
2208789.88176878715999.5906976412208798.61897581715926.416588794
 2208919.8477233715673.0375850262208934.04568472715574.744005978
#Sta/Elev= 30
       0 1569.01    11.4 1561.83    25.8 1556.68    46.7 1551.55    54.8 1550.18
    75.1 1547.31    90.8 1546.67    93.8 1545.78  100.211542.249   106.1 1540.43
   108.8 1540.42     115 1540.62   120.81542.227   123.8  1543.6   128.3 1544.02
   163.8 1543.53   183.8 1544.61   225.6 1545.31   274.6 1544.46   314.5 1547.29
   318.9 1549.24   327.8 1555.66   345.6 1563.08   366.6 1568.37   374.6 1569.61
   382.7 1572.41   415.1 1590.89   427.2 1599.41   439.3 1606.57   453.9 1613.87
#Mann= 6 ,-1,0
       0     .06       0  100.21    .045       0   120.8      .1       0
  303.69     .05       0  323.69     .06       0  424.58      .1       0
Bank Sta=100.21,120.8
XS Rating Curve= 0 ,0
Exp/Cntr(USF)=0,0
Exp/Cntr=0.3,0.1

Type RM Length L Ch R = 1 ,35918   ,34,32,31.9
XS GIS Cut Line= 3
2208912.78545585716090.5000229452209003.01896141 715681.79532127
2209004.78824583715587.138604649
#Sta/Elev= 30
       0 1576.08    17.7 1567.52      30 1567.94    62.8 1564.96    75.1 1559.44
    87.8 1555.58    91.5 1554.88   107.9 1554.53   120.1 1550.32   132.4 1547.74
   144.7 1544.03   185.7 1541.43  192.081540.011     198  1538.5   205.3 1538.42
   212.8 1539.94   218.7 1542.26   230.7 1543.61     284 1543.99   304.5 1542.89
   336.1 1543.16   346.2  1543.5   361.8 1545.44   382.3 1551.98   398.7  1559.6
   423.2 1566.47   459.2 1579.71   487.1 1592.06   499.2 1598.96   513.2 1608.11
#Mann= 6 ,-1,0
       0     .06       0      90      .1       0  192.08    .045       0
   212.8      .1       0     300     .05       0     380      .1       0
Bank Sta=192.08,212.8
XS Rating Curve= 0 ,0
Exp/Cntr(USF)=0,0
Exp/Cntr=0.3,0.1

Type RM Length L Ch R = 1 ,35886   ,74,83.5,87.9
XS GIS Cut Line= 3
2208944.63257546716098.4618028482209033.98143881 715681.79532127
2209034.86608102 715594.21574234
#Sta/Elev= 30
       0 1574.42     5.4 1569.95    17.7 1564.79    29.9 1566.17    46.3 1565.27
    58.6 1564.04    81.5 1559.26    95.4 1558.64    99.5 1557.35   115.2 1547.59
   128.1    1544   173.1 1539.53   182.6 1539.54   192.7 1538.15   201.8 1538.02
   205.9 1538.36   208.51539.521     214 1541.86   218.1 1542.57   238.6  1542.5
   275.4 1543.99     300  1543.4   353.1 1543.11   369.5 1544.59   377.7 1546.22
   406.3 1558.23   446.8 1571.14   466.8  1578.5   478.8 1584.16   513.7 1603.85
#Mann= 6 ,-1,0
       0     .06       0     100      .1       0   182.6    .045       0
   208.5      .1       0     240     .05       0     300      .1       0
Bank Sta=182.6,208.5
XS Rating Curve= 0 ,0
Exp/Cntr(USF)=0,0
Exp/Cntr=0.3,0.1

Type RM Length L Ch R = 1 ,35802   ,92.7,127.8,138
XS GIS Cut Line= 4
2208960.60769608716068.5593188962209003.38455371716017.240890755
2209219.88937985715728.2938493182209177.03654337715547.616013081
#Sta/Elev= 30
       0 1565.62    40.9    1562    58.9 1561.58    61.7 1560.92    78.8 1548.68
    88.1 1544.03    93.1 1542.59   106.9 1541.65   115.11538.997   121.7 1537.57
   131.9  1537.3   146.9 1537.56   151.81538.473   161.5 1542.46   164.6 1542.74
   201.5 1540.72   234.9 1540.26   308.3 1543.09   350.3 1542.74   361.8  1544.9
     376 1542.69   386.8 1542.25   406.8 1543.52     416  1545.4   435.2 1546.98
     464 1552.81   488.6 1560.13   524.1  1569.5   556.5 1581.96   613.6 1607.65
#Mann= 9 ,-1,0
       0     .06       0      60      .1       0   86.81     .07       0
   115.1    .045       0   151.8     .07       0  206.81     .05       0
  216.81      .1       0  386.81     .05       0  457.87      .1       0
Bank Sta=115.1,151.8
XS Rating Curve= 0 ,0
Exp/Cntr(USF)=0,0
Exp/Cntr=0.3,0.1

Type RM Length L Ch R = 1 ,35675   ,103.3,92.1,98.2
XS GIS Cut Line= 6
2208965.86398853716072.8071787162209029.62015271716019.693260343
2209107.24104517716013.820413959 2209333.4168051715961.221400023
2209465.04195514715889.0641003172209672.69311545715932.149067101
#Sta/Elev= 30
       0 1565.28    63.9 1560.78    68.2 1559.13    81.1 1549.45    85.5 1547.64
   157.7 1543.83   172.2 1541.31   182.3 1537.92   198.9 1534.35   214.5 1534.26
   223.3 1535.14  230.41 1537.94   243.8 1540.32   272.4 1539.12   329.8 1541.03
   377.5 1538.77   387.7 1540.11   452.1 1542.22   473.4 1541.15   544.7 1541.73
   551.4 1542.96   577.3 1552.22   611.1 1555.01   634.8  1554.6     645 1557.87
   657.6 1565.75   669.8 1570.96   682.1 1582.22   692.3 1589.04   756.2 1620.75
#Mann= 7 ,-1,0
       0     .06       0      40      .1       0   182.3    .045       0
  230.41     .07       0  523.29     .05       0  574.09     .06       0
  634.09     .07       0
#XS Ineff= 2 , 0
                          327.43         1548.18
Permanent Ineff=
       F       F
Bank Sta=182.3,230.41
XS Rating Curve= 0 ,0
Exp/Cntr(USF)=0,0
Exp/Cntr=0.3,0.1

Type RM Length L Ch R = 1 ,35583   ,159.2,148.3,123.8
XS GIS Cut Line= 6
2208966.85248815716163.5508684892209030.60865233716110.436950116
2209108.22954479716104.5641037332209334.40530472716051.965089796
2209466.03045476715979.8077900912209673.68161507716022.892756874
#Sta/Elev= 30
       0 1589.66    43.4 1576.22    53.8 1570.17    78.7 1559.28   128.7 1553.09
   140.7 1549.74   164.9 1546.33   223.7 1541.28   230.4 1540.02   236.71537.474
   242.8 1535.22     251 1534.48   267.6 1535.22   284.51538.397   312.3 1539.44
   324.6 1538.58   399.3 1538.87   464.1 1542.28     503 1543.05   550.4 1547.01
   562.6 1553.67   566.7 1554.59   603.5 1556.49   619.8 1562.05   632.7 1570.67
   652.5 1576.68   681.1 1594.92   693.4 1600.71   721.9 1617.42   756.2 1635.05
#Mann= 4 ,-1,0
       0      .1       0   236.7    .045       0   284.5      .1       0
  503.29     .07       0
#XS Ineff= 2 , 0
                          478.92         1549.38
Permanent Ineff=
       F       F
Bank Sta=236.7,284.5
XS Rating Curve= 0 ,0
Exp/Cntr(USF)=0,0
Exp/Cntr=0.3,0.1

Type RM Length L Ch R = 1 ,35434   ,517.4,529.7,541.4
XS GIS Cut Line= 5
2208986.12287491716278.8300853622209138.31864886716200.533344259
2209293.75318423716190.258145359 2209380.9046795716107.844804342
2209681.15243014 716123.40614303
#Sta/Elev= 30
       0 1606.52    47.3 1591.02      91 1573.42   168.7 1547.12     189 1544.67
   217.1 1543.61   335.8  1542.6   340.7 1541.54   346.4 1535.24   348.51534.104
   363.3 1532.53   371.8 1533.72   374.3 1535.28   379.8 1541.09   385.3 1541.78
   436.9 1541.15   445.9 1543.04   454.2 1541.33   470.3 1541.19   494.2 1542.89
   498.2 1543.83   510.2 1551.39   518.2 1555.12   550.3 1557.16   557.9 1558.74
   578.3 1567.65   610.4 1576.04   666.4 1599.53   714.5    1627   747.5 1643.48
#Mann= 7 ,-1,0
       0      .1       0  326.93     .05       0   348.5    .045       0
   371.8     .05       0  456.88      .1       0  556.88     .06       0
  656.88      .1       0
Bank Sta=348.5,371.8
XS Rating Curve= 0 ,0
Exp/Cntr(USF)=0,0
Exp/Cntr=0.3,0.1
